HEC-RAS study LAURELFK.prj: LAURELFK

--- LAURELFK.g01 (geometry) --- (continued)

Type RM Length L Ch R = 1 ,159100  ,219.7,219.7,219.7
XS GIS Cut Line= 2
2341079.59258527636526.5488659422341556.85078958636041.132401726
#Sta/Elev= 30
       0 3150.76    26.8  3139.8      41 3136.13    52.2 3131.62      58 3130.38
    92.1 3118.44     106 3114.41   120.6 3108.21   137.1 3106.89     159 3106.46
   170.2 3107.65   183.4  3105.4   194.8 3105.07   369.1 3106.07     420  3104.9
   439.5 3104.89   448.3 3102.09   470.9 3101.11   485.1 3101.12   494.73102.044
   502.9 3103.32   510.5 3107.09   531.4 3122.69   564.3 3135.03   594.2 3149.29
     617 3158.84   635.8 3169.46     647  3174.4   662.7 3183.32   680.7 3195.84
#Mann= 5 ,-1,0
       0      .1       0     280     .06       0     420      .1       0
   448.3    .045       0   494.7      .1       0
#XS Ineff= 2 , 0
          324.08 3118.59
Permanent Ineff=
       F       F
Bank Sta=448.3,494.7
XS Rating Curve= 0 ,0
Exp/Cntr(USF)=0,0
Exp/Cntr=0.3,0.1

Type RM Length L Ch R = 1 ,158880  ,37.8,37.8,37.8
XS GIS Cut Line= 5
2341031.85837676636600.6432871552341485.63912515636378.531375229
2341604.19423984636342.654192821 2341698.3903109 636286.76592379
2341810.56638456636168.471155199
#Sta/Elev= 30
       0 3185.64    44.9 3164.82    53.7 3163.36    62.6 3157.86    89.5 3146.05
     134 3133.24   155.3 3131.62   178.5  3127.3   196.3 3121.86   212.1 3110.03
   218.6 3107.49   362.7 3103.79   472.3 3105.95     507 3103.46   537.1 3104.24
  550.57 3100.41   569.3 3098.72  588.21 3100.41   601.4 3105.13   612.4 3106.42
   629.1 3106.34     643 3103.34   653.5 3104.38   680.2 3120.24   738.6 3136.45
   779.4 3151.85     840 3178.47     857 3189.41   869.1 3193.05   901.6 3212.03
#Mann= 7 ,-1,0
       0      .1       0     290     .06       0     400     .07       0
  505.22     .06       0  550.57    .045       0  588.21     .06       0
  659.09      .1       0
#XS Ineff= 2 , 0
                          624.93         3113.24
Permanent Ineff=
       F       F
Bank Sta=550.57,588.21
XS Rating Curve= 0 ,0
Exp/Cntr(USF)=0,0
Exp/Cntr=0.3,0.1

Type RM Length L Ch R = 1 ,158843  ,166.6,166.6,166.6
XS GIS Cut Line= 5
2341038.86781772636637.6573649832341492.64856612636415.545453058
2341611.20368081 636379.668270652341705.39975186636323.780001619
    2341841.7601636180.664530276
#Sta/Elev= 30
       0  3185.7    14.8 3181.85    64.1 3161.17   108.3 3144.96   129.9 3140.15
   152.9 3137.08   215.2 3114.72   237.5 3109.57   294.4  3104.6   446.8 3102.34
   469.1 3103.68   550.7 3101.48   559.1 3099.87   586.9 3098.49  600.01 3099.84
     605 3102.43   622.2 3106.16   663.7 3107.22   681.2 3105.66   698.8 3114.99
   756.6 3131.27   794.8 3146.48   806.4 3149.82     814 3153.77   824.5 3156.36
   841.2 3165.56   852.8 3169.33   869.3 3179.16   891.4 3188.84   936.3 3212.98
#Mann= 7 ,-1,0
       0      .1       0     280     .06       0     480     .07       0
     500     .06       0   559.1    .045       0  600.01     .06       0
  729.09      .1       0
Bank Sta=559.1,600.01
XS Rating Curve= 0 ,0
Exp/Cntr(USF)=0,0
Exp/Cntr=0.3,0.1

Type RM Length L Ch R = 1 ,158676  ,163.2,163.2,163.2
XS GIS Cut Line= 3
2341091.13153794636780.9340548452341628.28988026636542.973161992
2341845.87237022636261.598505848
#Sta/Elev= 30
       0 3174.33    44.9 3168.39   103.7 3166.75   140.1 3164.23   197.7 3151.49
   254.9  3141.1   276.8 3135.47   288.6    3127   297.7 3122.24   316.1 3121.79
     338 3106.15   346.2 3102.16   354.9 3100.38   368.6 3101.53   438.6 3101.53
   512.9 3098.13   534.9 3098.31   565.5 3097.32  576.46  3098.3     583 3101.39
   587.4 3101.78   652.7  3100.5   751.6 3101.27   768.3 3108.32     792 3109.85
   807.2 3118.94   837.5  3126.6   859.6 3134.27   914.3 3158.19   943.2 3173.09
#Mann= 10 ,-1,0
       0      .1       0     220     .06       0     380     .07       0
     440      .1       0   534.9    .045       0  576.46      .1       0
  607.51     .06       0  677.51     .07       0  737.51     .06       0
  857.51      .1       0
Bank Sta=534.9,576.46
XS Rating Curve= 0 ,0
Exp/Cntr=0.3,0.1

Type RM Length L Ch R = 1 ,158513  ,261.8,261.8,261.8
XS GIS Cut Line= 2
2341497.53086158636874.1130108652341938.87801433636340.658626235
#Sta/Elev= 30
       0 3194.77    11.6 3187.15      22 3182.54    28.1 3181.38    42.3 3173.37
    59.4 3165.52    79.2 3155.07    87.8  3152.5    99.9 3147.05   104.8  3144.4
   115.4  3136.8   133.2 3136.35   138.9    3135   150.3 3127.97     173 3116.46
   182.9 3110.36   195.7 3100.62   204.9 3096.15   223.8 3095.38   231.93096.098
   250.4 3098.34   323.1 3097.58   505.4 3100.15     548 3104.82   568.9 3108.04
   582.7 3112.71   603.4 3113.17   639.8 3125.56   669.3  3138.7   692.4 3151.14
#Mann= 8 ,-1,0
       0      .1       0      70     .06       0     200      .1       0
   204.9    .045       0   231.9      .1       0     330     .06       0
     450     .07       0     580     .06       0
Bank Sta=204.9,231.9
XS Rating Curve= 0 ,0
Exp/Cntr(USF)=0,0
Exp/Cntr=0.3,0.1

Type RM Length L Ch R = 1 ,158251  ,201.4,201.4,201.4
XS GIS Cut Line= 2
2341805.63276685636972.928314115 2342086.8470212636308.525639678
#Sta/Elev= 30
       0 3188.88    20.1 3179.08    38.4 3168.35    53.6 3156.01    56.2 3154.91
    73.6 3153.99    86.6 3144.76   108.6 3134.63   121.3 3127.59     133 3123.65
   160.5 3109.36   173.5 3096.23   177.8 3093.87   199.5 3093.88   209.3 3092.74
   230.6 3093.82   239.8 3095.64   442.8 3097.84   512.3 3106.78     547  3113.4
   555.7 3117.11   573.1 3117.88   612.1 3138.32   625.2 3143.52   642.6  3152.7
   651.8 3156.53   681.7 3173.94     699 3183.16   707.7 3186.47   721.5 3194.93
#Mann= 10 ,-1,0
       0     .06       0      60      .1       0     170     .06       0
     190      .1       0   199.5    .045       0   230.6      .1       0
     270     .06       0     380      .1       0     450     .06       0
     700      .1       0
Bank Sta=199.5,230.6
XS Rating Curve= 0 ,0
Exp/Cntr=0.3,0.1

Type RM Length L Ch R = 1 ,158050  ,250.3,250.3,250.3
XS GIS Cut Line= 2
 2341988.7694316637023.7872626672342303.46914052636405.901248816
#Sta/Elev= 30
       0 3171.75     7.4 3167.47    22.3 3166.59    43.3 3151.24    74.7 3135.36
    86.8 3132.06   102.6 3123.59   128.6 3114.46   142.1  3105.8   155.6 3093.45
   159.1 3091.86     177  3091.4     196 3091.87   272.3 3094.47   303.7 3092.51
   312.7 3093.87   326.1 3092.12   344.1 3095.39   357.6 3094.09   411.4 3095.52
   439.4 3093.93   448.2 3094.71   462.5 3099.09   501.2 3102.34   530.9 3110.23
   550.6 3117.45   559.6 3122.82   580.4  3124.6   599.3 3136.81   693.4  3180.9
#Mann= 8 ,-1,0
       0     .06       0     120      .1       0   159.1    .045       0
     196      .1       0     230     .06       0     340      .1       0
     450     .06       0     630      .1       0
Bank Sta=159.1,196
XS Rating Curve= 0 ,0
Exp/Cntr(USF)=0,0
Exp/Cntr=0.3,0.1

Type RM Length L Ch R = 1 ,157799  ,223.1,223.1,223.1
XS GIS Cut Line= 2
2342214.44250869637156.1035799082342556.11955108636382.453025011
#Sta/Elev= 30
       0 3164.48    77.5 3130.43   169.4 3102.15   173.7 3100.29   182.5 3092.75
   191.2 3089.56   208.7 3088.97   239.3 3089.59   248.1 3090.88   264.4 3089.13
   287.4 3089.61   326.8 3092.73   357.4 3091.05   383.6 3094.09   405.5  3093.2
   444.8 3094.73   501.7 3100.32     541 3102.02   562.9 3106.82   580.4 3115.35
   597.9 3116.39   619.8 3130.44   632.9 3133.31   663.5 3147.43     681 3152.63
   716.3 3168.06   746.6 3175.81   783.1  3180.1   828.6 3170.96   845.7 3165.67
#Mann= 8 ,-1,0
       0     .06       0      50      .1       0   191.2    .045       0
   239.3      .1       0     260     .06       0     370      .1       0
     480     .06       0     690      .1       0
#XS Ineff= 2 , 0
                          379.19         3107.46
Permanent Ineff=
       F       F
Bank Sta=191.2,239.3
XS Rating Curve= 0 ,0
Exp/Cntr=0.3,0.1

Type RM Length L Ch R = 1 ,157576  ,250.1,250.1,250.1
XS GIS Cut Line= 2
2342372.54956442 637238.704137052342760.16749858636693.736348436
#Sta/Elev= 30
       0 3156.11     6.6 3154.06    33.9 3140.46      51 3130.14    75.3 3121.42
    85.3 3115.74    98.4 3111.28   109.9 3104.99   129.5  3097.7   139.3 3096.34
     154 3091.07   167.2 3089.99   175.8 3086.82   193.3 3087.99   203.1 3086.69
   210.2 3086.36   238.9 3086.62   337.5 3093.25   351.3    3092   379.5 3095.37
   408.1 3094.67   461.7 3100.13   468.6 3101.28   482.4 3106.26     510 3107.91
   541.8 3109.44   580.2 3107.95   594.6  3108.8   603.2 3107.64   668.8 3111.33
#Mann= 7 ,-1,0
       0      .1       0   203.1    .045       0   238.9      .1       0
     340     .06       0     390      .1       0     510     .06       0
     630      .1       0
Bank Sta=203.1,238.9
XS Rating Curve= 0 ,0
Exp/Cntr(USF)=0,0
Exp/Cntr=0.3,0.1

Type RM Length L Ch R = 1 ,157326  ,236.6,236.6,236.6
XS GIS Cut Line= 3
 2342555.8375483637356.5398690452342799.77723241637104.751468072
  2343283.932347636701.128785577
#Sta/Elev= 30
       0 3146.74      12 3142.75    30.9 3131.37    69.5 3112.39   138.5 3098.42
   172.9 3087.39   195.9 3084.99   218.9 3085.08   237.4 3086.94   293.7 3083.81
   305.4 3083.94   319.4 3087.55   344.4 3086.55   364.8 3088.77   406.1 3088.28
   434.4 3098.51     450 3100.07   559.4 3100.99   586.3 3105.53   606.2  3105.8
   614.7 3111.04     626  3112.7   640.2    3118   649.8 3118.62   668.6 3126.58
   788.5 3158.38   845.8 3160.87   880.9 3157.89   944.8 3145.45   980.9 3141.26
#Mann= 7 ,-1,0
       0      .1       0   195.9    .045       0   218.9      .1       0
     310     .06       0  440.58      .1       0  570.58     .06       0
  690.58      .1       0
#XS Ineff= 2 , 0
                           355.7         3099.38
Permanent Ineff=
       F       F
Bank Sta=195.9,218.9
XS Rating Curve= 0 ,0
Exp/Cntr=0.3,0.1

Type RM Length L Ch R = 1 ,157090  ,295,295,295
XS GIS Cut Line= 2
2342735.99576427637484.6360489112343342.82929408636970.967832809
#Sta/Elev= 30
       0 3140.84    67.3 3114.44    84.1  3110.2   120.8 3097.89     136 3087.08
   141.6 3084.31   160.1 3083.04   194.1 3081.98   203.5  3083.1   212.6 3085.15
   235.3 3084.31   251.8 3081.89   272.7 3081.81     299 3084.78   311.9 3084.77
   321.1 3082.44   340.3 3081.39   356.6  3083.7   377.6 3082.32   389.2 3085.88
     430 3087.48   463.5 3086.09   502.1 3087.79     513 3085.86   531.6 3087.24
   562.6 3086.92   686.6  3090.5   707.7 3089.65   723.4 3091.44     795 3091.71
#Mann= 6 ,-1,0
       0      .1       0   160.1    .045       0   203.5      .1       0
     300     .06       0     430      .1       0     720     .06       0
#XS Ineff= 2 , 0
                           390.6         3104.97
Permanent Ineff=
       F       F
Bank Sta=160.1,203.5
XS Rating Curve= 0 ,0
Exp/Cntr(USF)=0,0
Exp/Cntr=0.3,0.1

Type RM Length L Ch R = 1 ,156795  ,247,247,247
XS GIS Cut Line= 3
2342871.86123079637695.033818315 2343408.6181457637416.710335496
2343630.37458104637335.543800324
#Sta/Elev= 30
       0 3143.57    16.4  3136.6    49.9 3124.85    63.4 3121.59   143.1 3095.95
   164.8 3083.66   179.6 3080.08   209.3 3078.22   224.2  3080.1   252.7  3081.5
   284.2 3079.86   356.3 3082.12   365.3  3080.8   387.8  3080.3   396.9 3085.49
   401.4 3086.52     420 3085.53   550.1 3086.22   581.6 3084.58   595.1 3085.79
   612.7 3083.43   642.5 3086.54   659.5 3085.63   685.1 3087.04     708  3093.3
   754.5 3108.76   787.3 3116.11   808.6 3123.28   821.4 3125.34   840.8 3131.02
#Mann= 5 ,-1,0
       0      .1       0   179.6    .045       0   224.2      .1       0
     330     .06       0     440      .1       0
#XS Ineff= 1 ,-1
   310.4  736.583103.816
Permanent Ineff=
       F
Bank Sta=179.6,224.2
XS Rating Curve= 0 ,0
Exp/Cntr=0.3,0.1

Type RM Length L Ch R = 1 ,156547  ,236.8,236.8,236.8
XS GIS Cut Line= 3
2342957.11681677637819.9043581032343112.12375492637832.141747957
2343666.88542831637677.134809804
#Sta/Elev= 30
       0 3133.64    19.4 3125.63    47.2 3111.35    55.2 3108.44    79.3 3093.61
    87.3 3091.63    99.4 3086.53   119.4 3082.57   155.5 3082.24   170.9 3078.31
   181.4 3079.46   197.1 3078.88   205.4 3077.31   238.6 3076.05   245.6  3077.3
   251.1 3079.28   263.5 3079.47   300.9 3077.88     330 3080.06   346.6  3082.8
   400.6 3081.09     492 3081.69   508.6 3080.16     541 3079.99   566.7 3081.96
   587.5 3081.91   595.8 3083.65     629 3095.51   683.8 3112.17   731.5 3124.34
#Mann= 5 ,-1,0
       0      .1       0   205.4    .045       0   245.6      .1       0
  315.49     .06       0  415.49      .1       0
#XS Ineff= 1 ,-1
  347.65  633.56 3100.17
Permanent Ineff=
       F
Bank Sta=205.4,245.6
XS Rating Curve= 0 ,0
Exp/Cntr(USF)=0,0
Exp/Cntr=0.3,0.1

Type RM Length L Ch R = 1 ,156311  ,241.8,241.8,241.8
XS GIS Cut Line= 4
2342767.88576596637926.4101505682343045.46312215638032.346780847
2343359.79671523638037.9422667752343620.17205073638035.462065478
#Sta/Elev= 30
       0 3155.46    81.7  3120.2    90.2 3117.78   104.6 3109.65   120.2 3104.18
   135.6 3095.04     163  3082.9   205.8  3077.5   244.1 3078.47   307.8 3077.41
   437.5 3080.77   451.8  3079.9   459.13075.791   483.8 3074.56   511.9 3075.76
   519.9 3077.11   539.9 3076.28   559.9 3079.28   611.9 3080.78   651.9  3077.9
   679.9 3078.91   699.9 3077.34   727.9 3078.97   759.9 3093.29   783.9 3096.83
   795.9 3100.34   819.9 3111.14   831.9 3115.23   847.9 3123.31   871.9 3131.84
#Mann= 5 ,-1,0
       0      .1       0   459.1    .045       0   511.9      .1       0
  607.11     .06       0  711.49      .1       0
Bank Sta=459.1,511.9
XS Rating Curve= 0 ,0
Exp/Cntr=0.3,0.1

Type RM Length L Ch R = 1 ,156069  ,302.4,302.4,302.4
XS GIS Cut Line= 3
 2342820.4659634638038.1378105032343116.20288487638117.680844555
2343479.24545055638360.389076663
#Sta/Elev= 30
       0 3107.75    20.4 3098.87    57.7 3085.57    67.5 3080.29    78.4 3077.56
   111.5 3076.45   132.2 3078.35   169.5 3075.49   210.9  3076.7   354.9 3077.31
   416.9 3079.88   463.7 3075.18   493.9 3076.75   527.5 3073.04   557.2 3072.59
     566 3073.06   571.2 3074.92     574 3077.31   585.3 3090.07   590.1 3094.03
   599.7 3098.66   614.8 3109.27   628.6 3115.55     643    3125   657.5  3131.2
   681.5 3143.93     696 3150.39   715.4 3162.33   729.6 3173.47   742.9 3181.26
#Mann= 5 ,-1,0
       0      .1       0  476.25     .06       0   527.5    .045       0
     566     .06       0  636.25      .1       0
Bank Sta=527.5,566
XS Rating Curve= 0 ,0
Exp/Cntr(USF)=0,0
Exp/Cntr=0.3,0.1

Type RM Length L Ch R = 1 ,155766  ,202.2,202.2,202.2
XS GIS Cut Line= 3
2342728.54966613638061.0031669372343110.56983306638455.387499189
2343170.21345003638530.602074194
#Sta/Elev= 30
       0 3130.39    33.8 3118.84    45.1 3112.88      57 3108.86    64.9 3104.71
     113 3083.99   135.6  3077.4   161.1 3076.88   175.2  3074.4   189.4  3073.6
   257.3 3073.86   278.7 3072.78   342.1 3074.63   356.3 3073.67   373.2 3074.65
   390.2 3073.79   430.6 3075.36   441.1  3074.8   452.5  3071.2   462.5 3070.27
   499.6 3071.13     507 3075.45   518.2 3077.73   523.2 3081.39   528.8 3087.54
   540.4 3098.12   564.5 3114.36   571.8 3118.79   585.7 3124.83   645.1 3160.19
#Mann= 4 ,-1,0
       0      .1       0   452.5    .045       0   499.6     .06       0
  609.07      .1       0
Bank Sta=452.5,499.6
XS Rating Curve= 0 ,0
Exp/Cntr=0.3,0.1

Type RM Length L Ch R = 1 ,155564  ,195,195,195
XS GIS Cut Line= 2
2342592.66697924638199.3138032122342998.34176864638610.584106954
#Sta/Elev= 30
       0 3126.07    15.1 3118.63    25.1 3114.68    33.5 3112.44    57.5  3100.2
      70 3098.52    84.7 3091.52    94.3 3088.29   111.3 3081.04   131.8 3074.19
   147.4 3073.07   175.9 3074.02   196.1 3075.82   210.1 3074.72   232.8  3070.5
   261.1 3072.94   289.2 3070.37   334.1 3072.72   345.3 3071.53   363.8 3072.64
   390.3 3071.23   422.4  3071.3   440.9 3072.05   457.7 3073.98   464.8 3080.72
   480.2 3093.22   500.5 3103.87   511.9 3111.36   546.1 3125.87   577.7 3142.39
#Mann= 4 ,-1,0
       0      .1       0   390.3    .045       0   422.4     .06       0
     560      .1       0
Bank Sta=390.3,422.4
XS Rating Curve= 0 ,0
Exp/Cntr(USF)=0,0
Exp/Cntr=0.3,0.1

Type RM Length L Ch R = 1 ,155369  ,297,297,297
XS GIS Cut Line= 3
2342414.69720403638398.2407774172342832.54831014638677.241740497
2342911.03797101638720.894258058
#Sta/Elev= 30
       0 3119.45    11.4 3113.47    55.1  3096.3    63.7 3091.94   124.3 3078.13
   127.7 3076.92   136.4 3069.85   146.1 3068.05   189.4 3070.85     207 3070.77
   228.6 3068.32   242.6  3070.8   251.9 3071.34   288.7 3070.94   303.1 3069.69
   323.3 3071.42   338.5  3069.1   376.9 3070.35   395.4 3069.61   415.9 3068.97
  430.98 3069.63   438.7 3072.34   453.9 3075.18   468.3 3081.33   477.9 3083.89
   487.7 3088.42   506.6 3094.74   538.6  3109.6   559.9 3116.76   592.2 3124.95
#Mann= 5 ,-1,0
       0      .1       0     360     .06       0   395.4    .045       0
  430.98     .06       0  542.44      .1       0
Bank Sta=395.4,430.98
XS Rating Curve= 0 ,0
Exp/Cntr=0.3,0.1

Type RM Length L Ch R = 1 ,155072  ,242.4,242.4,242.4
XS GIS Cut Line= 4
2342296.59324231638763.2913601692342661.56951265638801.519185165
2342712.04596777638798.5499819222342874.17890338638802.279775261
#Sta/Elev= 30
       0 3119.99    11.6 3117.06    19.7 3114.01    35.8 3110.49    59.9 3103.63
      76 3097.74    92.1 3087.59   112.2 3073.12   120.2 3068.66   128.8  3067.9
   160.5 3068.84   176.5 3065.87   192.6    3066   214.73067.624   228.8 3065.66
   251.93066.216   289.2 3067.94   301.2 3069.48   325.4 3069.09   369.6 3070.72
   397.6 3069.97   441.7 3071.16   492.8 3069.02   505.7 3069.23   513.3 3070.69
   521.5 3073.63   545.7 3085.08   557.7 3087.14   566.5  3090.5   579.7 3093.96
#Mann= 5 ,-1,0
       0      .1       0   214.7    .045       0   251.9      .1       0
  477.54     .06       0  577.54      .1       0
Bank Sta=214.7,251.9
XS Rating Curve= 0 ,0
Exp/Cntr(USF)=0,0
Exp/Cntr=0.3,0.1

Type RM Length L Ch R = 1 ,154830  ,338.4,338.4,338.4
XS GIS Cut Line= 3
2342370.39096128639106.3075935542342665.19247701638951.683189812
2342942.34386948638836.856390037
#Sta/Elev= 30
       0 3157.31    29.1 3143.11    33.6 3139.91    47.2 3127.29    71.3 3109.36
    78.8 3104.22    92.4 3096.59   119.5 3076.56   128.5 3071.52   137.5 3064.49
     144  3063.8   191.7  3063.5   199.7 3064.41   206.6 3066.61   214.3 3066.72
   223.3 3064.08   227.9 3063.91   242.1 3067.81     273 3067.43   300.1 3068.58
   409.7 3067.45   457.4 3065.89     484  3068.7   514.6 3067.26     530 3068.81
   545.3 3072.01   565.6  3079.4   600.4 3087.02   613.2 3091.65   632.9 3096.79
#Mann= 5 ,-1,0
       0      .1       0   137.5    .045       0   199.7      .1       0
  442.89     .06       0  552.89      .1       0
#XS Ineff= 2 , 0
                          486.72         3076.46
Permanent Ineff=
       F       F
Bank Sta=137.5,199.7
XS Rating Curve= 0 ,0
Exp/Cntr=0.3,0.1

Type RM Length L Ch R = 1 ,154491  ,182.8,182.8,182.8
XS GIS Cut Line= 3
2342750.61147872639329.4956116532342866.89742646639012.023826513
2342936.10180294638849.903608818
#Sta/Elev= 30
       0 3138.14     4.6  3135.5    30.2 3124.75    68.5 3105.25   101.2 3091.12
   111.1 3084.16   123.9 3073.47   136.7 3065.05   145.2 3063.48   166.5 3063.42
   172.9 3061.44   179.3 3060.59   196.3 3060.47   230.4  3060.6  234.34 3061.43
   243.2 3063.58   247.4 3063.81   263.4 3062.69   302.8 3063.53   318.6 3066.24
     332  3065.4   349.9 3066.58   423.5 3066.94   445.6 3068.08   454.3 3069.61
   466.2 3073.08   480.4 3078.59   489.1 3080.73   497.8 3084.76   514.4 3090.76
#Mann= 5 ,-1,0
       0      .1       0   172.9    .045       0  234.34      .1       0
     330     .06       0   478.1      .1       0
Bank Sta=172.9,234.34
XS Rating Curve= 0 ,0
Exp/Cntr(USF)=0,0
Exp/Cntr=0.3,0.1

Type RM Length L Ch R = 1 ,154309  ,286.4,286.4,286.4
XS GIS Cut Line= 3
2342884.46316694639454.8797604912343034.86881451639087.108630651
2343158.77563552638782.652703223
#Sta/Elev= 30
       0 3164.22    32.1 3149.43    62.3 3139.23   101.2 3120.24   135.8 3098.96
   191.2 3073.05   226.6 3062.41   256.8 3059.95   269.8 3061.51   283.3 3059.66
   308.7 3058.84  334.88 3059.65   353.8    3062   382.1 3060.63   402.9 3064.16
   427.4 3065.19   520.3 3064.17   550.6 3066.48   562.5 3068.72   576.5 3074.28
   589.4 3076.98   615.4 3092.05   619.7 3094.03   628.3 3095.08   654.2  3110.8
   662.9 3111.59   701.7 3131.58   710.4 3137.21     719 3139.88     726 3143.88
#Mann= 5 ,-1,0
       0      .1       0   283.3    .045       0  334.88      .1       0
  397.34     .06       0  507.34      .1       0
Bank Sta=283.3,334.88
XS Rating Curve= 0 ,0
Exp/Cntr=0.3,0.1

Type RM Length L Ch R = 1 ,154022  ,241.3,241.3,241.3
XS GIS Cut Line= 2
2343196.22168504 639413.371722092343363.46601305638885.124393385
#Sta/Elev= 30
       0 3099.49    16.1 3095.82    33.8 3088.75    42.2 3084.03    54.7 3074.98
    84.1 3059.41    88.3 3058.25   100.9 3059.66   121.2 3057.61   155.4  3059.3
     210 3057.96     220  3057.2   235.2 3058.64   243.6 3057.74   264.5 3056.75
   293.9  3057.7   298.1 3058.63     306 3062.94   310.7 3063.37   340.1 3059.59
   365.2 3060.47   386.2 3063.42   407.2 3064.78   440.7 3063.02   474.3 3064.48
   494.1 3069.14   507.9 3076.37   520.5 3078.92   529.1 3084.69   554.1 3097.14
#Mann= 7 ,-1,0
       0      .1       0     210     .08       0     240      .1       0
   243.6    .045       0   293.9      .1       0     350     .06       0
     450      .1       0
Bank Sta=243.6,293.9
XS Rating Curve= 0 ,0
Exp/Cntr(USF)=0,0
Exp/Cntr=0.3,0.1

Type RM Length L Ch R = 1 ,153781  ,250.3,250.3,250.3
XS GIS Cut Line= 2
2343447.56764976639530.6415364842343575.74028214638887.979508686
#Sta/Elev= 30
       0 3142.52    74.9  3102.1   103.5 3073.11   119.8 3061.32   127.9 3057.86
   144.2 3055.18   156.5 3057.47   193.2 3058.94   213.6 3054.96     250 3058.56
   258.5 3055.44   290.8  3057.3   303.3 3056.02   319.6  3054.8   333.63055.863
   344.1 3060.47   364.5 3056.48   409.4 3062.12   450.2 3061.92   458.3  3060.7
   470.6 3062.14   503.2 3060.61   527.7 3062.48   539.9 3061.81   552.7  3063.7
   573.1 3068.75   610.5 3084.57   625.5 3087.87   633.7 3093.68   655.3 3104.41
#Mann= 5 ,-1,0
       0      .1       0   303.3    .045       0   333.6      .1       0
     360     .06       0     540      .1       0
Bank Sta=303.3,333.6
XS Rating Curve= 0 ,0
Exp/Cntr=0.3,0.1

Type RM Length L Ch R = 1 ,153530  ,246.2,246.2,246.2
XS GIS Cut Line= 2
2343638.44032572639538.9902437122343868.70840542638974.833448456
#Sta/Elev= 30
       0 3118.24     8.9 3114.68    39.5 3099.29    75.4 3085.15    85.6 3079.07
     107 3062.43   114.3 3057.99   127.2 3054.65   174.8 3052.96   186.8 3053.65
     196 3055.77   209.3 3056.25   237.5 3055.31   278.5 3055.59   300.3 3054.62
   330.3 3053.48  340.96 3054.65   351.9  3056.5     374 3055.17   389.3 3058.91
   404.6 3059.81     434 3057.68   447.6 3057.85   464.2 3059.17   481.5 3061.85
   521.2 3074.82   559.3 3090.04   567.9  3090.7   576.8 3094.75   609.3 3102.99
#Mann= 6 ,-1,0
       0      .1       0     170     .08       0     280     .06       0
   300.3    .045       0  340.96     .06       0     490      .1       0
#XS Ineff= 2 , 0
                           404.8         3067.41
Permanent Ineff=
       F       F
Bank Sta=300.3,340.96
XS Rating Curve= 0 ,0
Exp/Cntr(USF)=0,0
Exp/Cntr=0.3,0.1

Type RM Length L Ch R = 1 ,153284  ,268.3,268.3,268.3
XS GIS Cut Line= 2
2343698.17624878639607.1477963872344209.87757679639162.571677554
#Sta/Elev= 30
       0 3134.79    27.4 3121.44    39.7 3113.68    50.3 3108.47    92.7 3091.77
   112.8  3081.8   149.4 3070.02   187.1 3052.42   192.1  3051.8   204.1 3053.59
   235.3 3054.26   300.5 3051.33   331.2 3050.67   348.7 3051.35   371.4 3054.83
   393.3 3056.18   419.6 3055.23   445.1 3056.84   484.8 3057.16     506 3056.29
   521.7 3053.56   537.8 3053.96   552.9 3056.66   564.2 3062.02   576.3  3069.6
   603.9 3080.23   635.1 3088.18   643.8 3092.19   660.6 3094.79   677.9  3100.6
#Mann= 5 ,-1,0
       0      .1       0   300.5    .045       0   348.7      .1       0
     460     .06       0     590      .1       0
#XS Ineff= 2 , 0
                          393.73         3064.75
Permanent Ineff=
       F       F
Bank Sta=300.5,348.7
XS Rating Curve= 0 ,0
Exp/Cntr=0.3,0.1

Type RM Length L Ch R = 1 ,153016  ,220.2,220.2,220.2
XS GIS Cut Line= 2
2343818.81698815639834.5009459882344382.97378341639366.289183939
#Sta/Elev= 30
       0 3154.47    30.3 3140.37   100.5 3113.94   115.5 3105.65   158.1 3087.68
   180.9 3079.32   235.7 3062.04   252.6 3054.95  263.03 3048.97   268.9 3048.16
   340.3 3048.95   368.3 3050.08   402.9 3048.81   416.6  3050.3     428 3054.28
   440.5  3055.3   476.3 3055.24   516.4 3051.62     547 3052.99     572 3050.44
   603.3 3053.12   612.6 3051.37   632.5 3051.42   646.7 3054.27   660.9 3061.49
   672.2 3069.12     691 3077.82   709.2 3082.32   719.1 3086.07   733.1 3087.21
#Mann= 5 ,-1,0
       0      .1       0  263.03    .045       0   340.3      .1       0
     550     .06       0     680      .1       0
#XS Ineff= 2 , 0
                          472.13         3062.46
Permanent Ineff=
       F       F
Bank Sta=263.03,340.3
XS Rating Curve= 0 ,0
Exp/Cntr(USF)=0,0
Exp/Cntr=0.3,0.1

Type RM Length L Ch R = 1 ,152796  ,249.1,249.1,249.1
XS GIS Cut Line= 2
2343905.14593128 639960.442517182344530.67924554639638.901785577
#Sta/Elev= 30
       0 3146.89    16.9 3142.15    37.3 3132.94    88.9 3114.58   138.3 3091.87
   156.2 3085.51   174.3 3076.21   184.6 3072.68   219.3 3056.27   230.4 3053.97
   241.8 3053.49   250.8 3049.23   257.2 3047.83   291.2 3046.66  315.01 3047.84
   327.2 3050.23   358.7 3050.28   394.7 3049.96   414.6 3047.92   475.6 3047.88
   493.6 3050.32   530.5 3051.92   543.1 3049.41   556.6 3053.14   570.1 3052.54
   583.9 3061.91   592.8 3065.48   645.9  3074.8     678 3082.58   703.3 3086.26
#Mann= 5 ,-1,0
       0      .1       0   257.2    .045       0  315.01      .1       0
     410     .06       0     600      .1       0
#XS Ineff= 2 , 0
                          522.15         3064.74
Permanent Ineff=
       F       F
Bank Sta=257.2,315.01
XS Rating Curve= 0 ,0
Exp/Cntr=0.3,0.1

Type RM Length L Ch R = 1 ,152547  ,248.9,248.9,248.9
XS GIS Cut Line= 2
2344016.38446737640142.1609544562344565.57383745639928.011640338
#Sta/Elev= 30
       0 3108.16      47 3088.44    72.8 3076.56    85.6 3072.84   102.8 3063.21
   115.7 3059.77   128.6 3054.74   142.7 3051.04     150 3048.23   158.6 3047.65
   164.3 3046.02   167.4 3045.15   232.3 3046.04   240.2 3048.09   318.8 3048.33
   346.6 3046.89   355.8 3048.04   389.8    3047   424.8 3048.06     442 3047.79
   451.6 3044.84   465.1 3044.16   476.3 3045.28   488.6 3050.66   497.9 3051.29
   507.2  3054.6   538.1 3059.85   565.9  3066.5   575.1 3069.67   589.5 3072.24
#Mann= 5 ,-1,0
       0      .1       0   164.3    .045       0   232.3      .1       0
     460     .06       0     560      .1       0
Bank Sta=164.3,232.3
XS Rating Curve= 0 ,0
Exp/Cntr(USF)=0,0
Exp/Cntr=0.3,0.1

Type RM Length L Ch R = 1 ,152298  ,201.1,201.1,201.1
XS GIS Cut Line= 3
2343999.33361558640427.8513996442344393.43577239640244.754128139
2344637.23085663640113.199057346
#Sta/Elev= 30
       0 3110.22    75.9 3078.04     102 3068.31   132.1 3059.62   159.7 3054.47
   198.4 3050.07     217 3049.39   239.1  3046.2   283.2 3048.73   306.8 3044.03
   342.9 3044.07     349 3044.61   358.2 3043.18   375.8  3046.6   397.9 3044.56
   442.1 3046.75   455.9 3044.76   501.3 3042.01   527.8 3043.09   542.5 3045.76
     560  3041.4   587.7 3044.23   605.8 3049.47   614.9 3056.82   628.6 3064.25
   655.8 3072.52   669.4 3079.48   687.7 3081.37   701.3  3089.9   711.6 3093.94
#Mann= 5 ,-1,0
       0      .1       0   306.8    .045       0   342.9      .1       0
  494.56     .06       0  604.56      .1       0
#XS Ineff= 2 , 0
          279.19 3056.17
Permanent Ineff=
       F       F
Bank Sta=306.8,342.9
XS Rating Curve= 0 ,0
Exp/Cntr=0.3,0.1

Type RM Length L Ch R = 1 ,152097  ,311,311,311
XS GIS Cut Line= 2
2344064.74076411640622.2699006222344665.74045211640314.862014228
#Sta/Elev= 30
       0  3082.4    39.8  3072.3    97.4 3061.45   134.2  3048.5   143.1 3046.88
   165.6 3045.98   197.1  3047.6   244.1 3047.39   264.4 3045.66   268.9 3042.95
   277.9 3041.84  312.04 3042.94   327.4 3045.03   349.8 3041.49   372.3 3043.68
   426.2 3040.93   441.6 3043.21   457.6 3042.88   471.1 3044.53   489.1 3041.56
   507.1 3040.48   529.5 3040.81     552 3047.11   556.5 3049.26     570 3061.49
   583.4 3070.83   610.4  3083.2   628.4 3087.14   641.8 3095.69   675.1 3111.44
#Mann= 5 ,-1,0
       0      .1       0   268.9    .045       0  312.04      .1       0
     530     .07       0     570      .1       0
Bank Sta=268.9,312.04
XS Rating Curve= 0 ,0
Exp/Cntr(USF)=0,0
Exp/Cntr=0.3,0.1

Type RM Length L Ch R = 1 ,151786  ,138.1,138.1,138.1
XS GIS Cut Line= 3
2344136.49550422640923.2159216472344410.05205073640763.172399351
2344690.59835187640588.410715234
#Sta/Elev= 30
       0 3086.72    87.7 3071.57   157.2 3047.87   173.8 3044.34   208.2 3042.77
   254.5 3045.25     279 3043.42   296.2 3039.03   314.8 3038.92   333.6 3040.02
   338.3 3041.33   360.6  3041.9   385.4 3039.26   401.2 3038.24   421.6 3039.26
   437.3 3041.34   470.2 3041.39   482.5 3038.97   489.1    3040   503.2 3038.61
   512.7 3042.69   522.1 3044.17     529 3047.83   549.3 3065.41   566.7 3075.42
   588.1 3084.94   592.8 3088.17   606.9 3091.87   616.3 3098.95   647.5  3117.4
#Mann= 6 ,-1,0
       0      .1       0   385.4    .045       0   421.6      .1       0
  466.93     .08       0  516.93     .07       0  586.93      .1       0
#XS Ineff= 2 , 0
          254.83 3052.04
Permanent Ineff=
       F       F
Bank Sta=385.4,421.6
XS Rating Curve= 0 ,0
Exp/Cntr=0.3,0.1

Type RM Length L Ch R = 1 ,151648  ,346.6,346.6,346.6
XS GIS Cut Line= 2
2344273.28426775641034.3552425782344758.22884359640683.081287001
#Sta/Elev= 30
       0  3076.4    77.7 3066.13   102.4 3058.68     132 3045.36   157.6 3039.72
   186.2 3039.69   206.3 3041.93   245.6 3042.24   250.5 3041.95   260.4 3038.99
   281.6 3039.61   297.9 3038.31   304.9 3037.23   326.6 3037.14  342.19 3038.31
   359.2 3039.76   383.9 3039.44   401.1 3037.81   406.8 3038.68   418.2 3042.93
   433.3 3042.63     444 3048.94   478.4 3060.53   502.4 3070.74   515.6  3077.9
   527.1 3080.63     537 3088.69   552.9 3098.41   566.6 3108.43   598.8 3124.83
#Mann= 4 ,-1,0
       0      .1       0   297.9    .045       0  342.19     .08       0
     450      .1       0
Bank Sta=297.9,342.19
XS Rating Curve= 0 ,0
Exp/Cntr(USF)=0,0
Exp/Cntr=0.3,0.1

Type RM Length L Ch R = 1 ,151301  ,255.3,255.3,255.3
XS GIS Cut Line= 4
 2344340.0837758641259.0998346852344597.42812217641082.704571091
2344784.18832363640909.3124313242344867.73361849640728.643169562
#Sta/Elev= 30
       0 3082.66    53.5  3072.6     131 3053.95   153.9 3052.64   168.3 3048.82
   188.5 3039.66   201.5 3036.74   232.9 3035.57   248.9 3036.75   266.8 3036.26
   286.2 3038.69   300.8 3037.81   321.2 3039.44   408.5 3040.53   456.5 3035.52
   473.5 3037.46   496.5 3037.29   513.1 3040.05   544.3  3038.1   558.4 3039.86
   571.4 3037.91   584.6 3040.52   611.1 3040.85   641.9 3043.53   666.4  3050.7
   699.2 3064.77   712.4 3067.34   738.3 3084.09   752.1 3088.01   765.9 3097.03
#Mann= 5 ,-1,0
       0      .1       0   201.5    .045       0   248.9      .1       0
     502     .07       0  626.84      .1       0
#XS Ineff= 2 , 0
                          524.53         3044.84
Permanent Ineff=
       F       F
Bank Sta=201.5,248.9
XS Rating Curve= 0 ,0
Exp/Cntr=0.3,0.1

Type RM Length L Ch R = 1 ,151046  ,285.8,285.8,285.8
XS GIS Cut Line= 3
2344686.73060484641463.3446750522344745.79436728641164.917243766
2344929.20289276640735.927811292
#Sta/Elev= 30
       0 3122.11    51.1 3098.22   100.1 3078.06   138.2    3051   153.4 3036.67
   159.7 3034.01   197.1 3033.22   213.5 3033.92   230.6 3037.22   308.3 3035.31
   321.3 3038.04   343.1 3038.59   369.2 3036.42     412 3037.75   443.1 3034.74
   462.9  3036.2   473.6 3040.47   543.2 3039.03   551.9 3037.38   561.8 3039.24
     578 3036.92     591 3037.92   617.1 3036.51   678.1 3048.29   695.5 3055.31
   704.2 3060.69   721.6 3063.55   730.3 3069.61   747.7 3078.58   770.8 3088.86
#Mann= 5 ,-1,0
       0      .1       0   159.7    .045       0   213.5      .1       0
  534.22     .06       0  644.22      .1       0
#XS Ineff= 2 , 0
                          519.16         3047.89
Permanent Ineff=
       F       F
Bank Sta=159.7,213.5
XS Rating Curve= 0 ,0
Exp/Cntr(USF)=0,0
Exp/Cntr=0.3,0.1

Type RM Length L Ch R = 1 ,150760  ,265.5,265.5,265.5
XS GIS Cut Line= 3
2345029.12107635641389.9486625372344990.73795261641179.332438916
2345010.05396261640734.873216956
#Sta/Elev= 30
       0 3094.98    61.8  3067.3    87.5 3052.68   106.5 3039.32   114.6 3034.64
   118.7 3033.59   143.1  3034.2   155.3 3031.59   204.1 3030.95   212.2 3031.53
   224.2 3034.66   296.3 3035.73   312.3 3038.46   324.3 3039.03   340.3 3038.22
   408.4  3038.9   432.4  3036.5   468.5 3037.28   480.5  3035.4   488.5 3038.01
   492.5 3038.16   507.8 3035.22   548.6 3038.83   584.6 3045.77   604.6 3055.51
   612.5 3056.21   616.6 3057.67   636.6 3070.94   648.6 3074.87     659 3079.91
#Mann= 5 ,-1,0
       0      .1       0   155.3    .045       0   212.2      .1       0
  444.09     .06       0  544.09      .1       0
#XS Ineff= 2 , 0
                          406.39         3044.33
Permanent Ineff=
       F       F
Bank Sta=155.3,212.2
XS Rating Curve= 0 ,0
Exp/Cntr=0.3,0.1

Type RM Length L Ch R = 1 ,150494  ,199.3,199.3,199.3
XS GIS Cut Line= 2
 2345282.3336518641312.5005904642345144.66301595640741.626353774
#Sta/Elev= 30
       0 3084.24    44.3 3065.28   106.3 3042.13   123.9 3030.08   130.5 3028.99
   163.7 3028.79   173.6    3030   180.3 3031.35   192.7 3031.17     205 3032.92
   221.5 3032.16   229.7 3030.69   242.1 3034.96   246.2 3035.35   269.8 3032.84
   286.3 3032.87   307.9    3035     356 3035.39   386.1 3037.24   447.8 3036.24
   460.1 3037.22   468.4 3035.62   501.3 3036.72   513.6  3039.3   521.9 3043.87
   534.2 3044.46   555.2 3052.95   567.1 3054.16   575.4 3059.45   587.2 3064.72
#Mann= 5 ,-1,0
       0      .1       0   123.9    .045       0   173.6      .1       0
     470     .06       0     570      .1       0
#XS Ineff= 2 , 0
                          320.15          3037.5
Permanent Ineff=
       F       F
Bank Sta=123.9,173.6
XS Rating Curve= 0 ,0
Exp/Cntr(USF)=0,0
Exp/Cntr=0.3,0.1

Type RM Length L Ch R = 1 ,150295  ,240.9,240.9,240.9
XS GIS Cut Line= 2
2345494.08613258 641289.228847812345275.41048566640606.030070793
#Sta/Elev= 30
       0 3105.05    12.7 3096.91    71.5 3065.53    88.3 3058.02   121.8 3045.67
   141.5 3040.01   155.4 3031.35   160.6 3029.67   176.3  3028.1   222.6 3029.56
     231 3031.09   252.9 3031.11   277.2 3029.29   289.8  3031.9   302.4 3031.47
   321.2 3035.69   352.8 3033.56   411.6 3034.85     420 3034.11   520.2 3035.47
     546 3037.56   567.9 3042.23     587 3048.73   596.4 3053.77     609 3056.44
   617.4 3062.39   634.7 3069.58   655.2 3080.92   680.4 3092.29   717.3 3110.87
#Mann= 5 ,-1,0
       0      .1       0   160.6    .045       0   222.6      .1       0
     460     .06       0     560      .1       0
Bank Sta=160.6,222.6
XS Rating Curve= 0 ,0
Exp/Cntr=0.3,0.1

Type RM Length L Ch R = 1 ,150054  ,244.3,244.3,244.3
XS GIS Cut Line= 3
2345695.34555938641244.5830767742345649.45534742640904.995508326
 2345592.5514846640581.928416179
#Sta/Elev= 30
       0 3091.37     7.5 3088.97    19.6 3082.34    27.7 3080.22    51.6  3067.6
   105.4 3046.75   156.8 3035.09   168.9 3027.97   188.13027.808   225.4 3026.67
   247.6 3027.94   286.8 3030.35   302.1 3029.31   334.4 3031.07     379  3029.5
   395.4 3026.75   399.3 3027.06   407.5 3031.61   415.6 3032.61   460.3 3030.22
   472.5 3032.75   488.7 3030.16   513.1 3030.38   545.6 3039.48   569.9 3051.17
   598.4  3061.6   618.7 3064.81   626.8 3069.06   634.9 3070.31   670.7  3080.7
#Mann= 5 ,-1,0
       0      .1       0   188.1    .045       0   247.6      .1       0
  392.67     .06       0  492.67      .1       0
#XS Ineff= 2 , 0
                          442.79         3041.94
Permanent Ineff=
       F       F
Bank Sta=188.1,247.6
XS Rating Curve= 0 ,0
Exp/Cntr(USF)=0,0
Exp/Cntr=0.3,0.1

Type RM Length L Ch R = 1 ,149810  ,520.6,520.6,520.6
XS GIS Cut Line= 3
2345929.38071409 641266.71457695     2345918.516641080.512682495
2345841.67961377640543.139967261
#Sta/Elev= 30
       0 3049.01    29.6 3042.22    57.6 3032.85    81.7 3026.94   141.8 3031.01
   193.9 3029.29   214.1 3030.62   239.53025.728   246.5 3024.81   294.9 3025.67
   331.3 3028.12   375.4 3025.83   389.5  3028.6   484.7 3028.03   505.1 3025.26
   525.3 3027.76   533.3 3026.92   545.5  3030.1   561.6 3028.88   577.8 3025.62
   585.9 3025.67     602 3030.42   626.4 3042.23   634.4 3046.75   650.5 3058.89
   670.7 3067.47   678.8 3070.04   690.9 3071.12     699 3076.51   729.4 3086.38
#Mann= 6 ,-1,0
       0     .06       0      20      .1       0   239.5    .045       0
   294.9      .1       0  516.52     .06       0  616.52      .1       0
#XS Ineff= 2 , 0
          211.65 3035.13
Permanent Ineff=
       F       F
Bank Sta=239.5,294.9
XS Rating Curve= 0 ,0
Exp/Cntr=0.3,0.1

Type RM Length L Ch R = 1 ,149289  ,293.8,293.8,293.8
XS GIS Cut Line= 3
2345919.26148039641358.0761860382346176.37325968640924.347332252
2346340.28371593640605.493749055
#Sta/Elev= 30
       0 3062.16    25.3    3056    88.9 3047.11   109.3 3041.78   131.2 3032.39
   150.8 3026.75   177.7 3025.93   196.3 3029.24   214.9 3027.58   252.4 3029.19
   349.8 3027.55   453.8 3029.72   489.3 3028.79   525.8 3024.36   561.7 3024.93
   570.83022.268   573.8  3021.9     6223022.917   637.1 3030.11   647.2 3029.61
   656.2 3032.91   669.7 3042.58   683.2 3056.02   701.2 3066.45   741.6 3082.07
   764.1 3088.76   785.6 3097.91   801.2 3099.63   818.3 3106.66   862.7 3119.37
#Mann= 7 ,-1,0
       0     .06       0     130      .1       0     190     .06       0
     380      .1       0   570.8    .045       0     622     .06       0
  694.21      .1       0
#XS Ineff= 2 , 0
          398.53 3039.72
Permanent Ineff=
       F       F
Bank Sta=570.8,622
XS Rating Curve= 0 ,0
Exp/Cntr=0.3,0.1

Type RM Length L Ch R = 1 ,148995  ,237.3,237.3,237.3
XS GIS Cut Line= 3
2345981.26908516641428.8501916732346323.91877524641061.745506803
2346580.49373737640931.281950342
#Sta/Elev= 30
       0 3046.95    33.6 3042.57    98.1 3037.94     166  3029.9   212.9 3027.04
   229.4    3025   251.2 3024.56     306 3028.35   338.8 3028.85   375.4 3025.56
   402.9 3026.83   420.9 3025.62   453.7 3026.62   470.1 3023.11   502.2 3025.99
   523.6 3025.53   565.3 3026.72   583.2 3023.72   591.7 3023.08   610.2 3023.87
   635.8 3020.37   645.6 3019.26     673 3019.31   684.1 3020.33   699.9 3026.54
   704.4  3029.2     717 3048.32   731.8 3063.58   767.2  3090.2     790    3105
#Mann= 6 ,-1,0
       0     .06       0     200      .1       0  602.17     .06       0
   635.8    .045       0   684.1     .06       0  732.17      .1       0
#XS Ineff= 2 , 0
          562.13 3052.16
Permanent Ineff=
       F       F
Bank Sta=635.8,684.1
XS Rating Curve= 0 ,0
Exp/Cntr(USF)=0,0
Exp/Cntr=0.3,0.1

Type RM Length L Ch R = 1 ,148758  ,208.3,208.3,208.3
XS GIS Cut Line= 3
2346015.21188778641468.2477034682346375.73519671641242.351406899
2346718.48652098641192.830037097
#Sta/Elev= 30
       0 3055.96    53.1 3051.89    81.3 3047.84   113.2 3033.15   141.4 3032.82
   208.8 3024.49   232.4 3024.11   254.4 3027.61   272.8 3027.75   310.5 3025.84
   331.6 3023.19   392.9 3021.17   442.1 3020.74     494 3022.57529.09523018.681
   539.1 3017.56   571.7 3018.65   579.5 3020.41   587.6 3028.31   591.6 3028.79
   599.7 3026.89   607.8 3029.29   628.2 3042.46   644.1 3057.61   648.2 3060.04
   696.7 3081.12     733 3099.22   741.3 3104.71   757.3 3109.03   771.8 3117.93
#Mann= 7 ,-1,0
       0      .1       0      40     .06       0     120      .1       0
  465.45     .06       0529.0952    .045       0   571.7     .06       0
  655.45      .1       0
#XS Ineff= 2 , 0
          494.29 3031.51
Permanent Ineff=
       F       F
Bank Sta=529.0952,571.7
XS Rating Curve= 0 ,0
Exp/Cntr=0.3,0.1

Type RM Length L Ch R = 1 ,148550  ,264.2,264.2,264.2
XS GIS Cut Line= 3
2346124.49884716641519.7092009632346383.31964257641442.613644883
2346697.20869232641396.723432931
#Sta/Elev= 30
       0 3050.59    28.9 3047.84    45.6 3047.16    95.7 3041.78   116.5 3036.92
     129 3032.79   141.6 3031.12   154.1 3026.47   158.3 3025.76   172.2 3026.59
   216.7  3024.4   241.7 3020.23   270.9 3018.42   287.1 3018.48   299.2 3021.64
   311.3 3022.19   319.4 3021.49   336.33018.202   343.7 3017.39   370.8 3017.05
   387.7 3018.09   416.5 3017.02   430.8  3019.2   456.9 3019.94     465 3022.38
   481.1 3021.71   504.9 3033.39   548.7 3059.93   557.8 3063.48   587.3 3080.16
#Mann= 5 ,-1,0
       0      .1       0   336.3    .045       0   387.7      .1       0
  400.06     .06       0  500.06      .1       0
#XS Ineff= 2 , 0
          258.72 3031.61  468.06         3027.89
Permanent Ineff=
       F       F
Bank Sta=336.3,387.7
XS Rating Curve= 0 ,0
Exp/Cntr(USF)=0,0
Exp/Cntr=0.3,0.1

Type RM Length L Ch R = 1 ,148286  ,224.9,224.9,224.9
XS GIS Cut Line= 3
2346122.45909538641779.8197138622346511.38893349  641664.7482044
2346775.04746471641577.345510837
#Sta/Elev= 30
       0 3044.26    26.8 3039.37    93.6 3033.78   139.4 3021.84   190.2  3021.3
     227 3023.55   268.8 3023.94   289.6 3021.76     298 3018.45   314.6 3018.17
   327.2 3015.08   360.5 3016.74   381.4 3015.42   406.4 3017.37   444.4 3016.27
     466 3015.09   478.1 3016.29   507.6    3020   520.2 3018.04   537.1 3018.43
   549.7 3021.83   583.1 3043.24   596.1 3052.91   604.5 3056.96   621.3  3069.8
     634 3075.65   642.4 3083.28   655.1 3087.06   667.7 3096.17   683.4 3104.45
#Mann= 5 ,-1,0
       0      .1       0     400     .06       0   444.4    .045       0
   478.1     .06       0   505.6      .1       0
#XS Ineff= 2 , 0
                          508.48         3026.98
Permanent Ineff=
       F       F
Bank Sta=444.4,478.1
XS Rating Curve= 0 ,0
Exp/Cntr=0.3,0.1

Type RM Length L Ch R = 1 ,148061  ,268.6,268.6,268.6
XS GIS Cut Line= 2
2346172.52455918641950.6924457522346775.52194423 641826.78887348
#Sta/Elev= 30
       0 3039.91    40.5 3030.52   130.3 3022.92   171.2 3017.64     211 3016.53
   231.3 3019.42   275.4 3015.74   289.6    3018   301.8 3015.66   314.1 3014.86
   338.6 3016.03   375.3 3015.62   385.83014.567   395.7  3013.1   424.2 3013.37
     438 3014.52   448.8 3017.01   469.3 3016.76   481.5 3018.24   489.7 3016.21
   505.7 3016.91   530.5 3015.44   538.7 3019.42   549.8 3027.25   559.9 3036.15
   575.4 3047.53   583.6  3054.9   599.9  3066.5     604 3068.66   615.6 3071.18
#Mann= 5 ,-1,0
       0      .1       0     340     .06       0   385.8    .045       0
     438     .06       0     440      .1       0
#XS Ineff= 2 , 0
          227.85 3030.21
Permanent Ineff=
       F       F
Bank Sta=385.8,438
XS Rating Curve= 0 ,0
Exp/Cntr(USF)=0,0
Exp/Cntr=0.3,0.1

Type RM Length L Ch R = 1 ,147792  ,243.3,243.3,243.3
XS GIS Cut Line= 3
2346174.37643371642179.1085499192346713.13239935      642106.409
2346879.04811945642070.832216045
#Sta/Elev= 30
       0 3057.97    66.4 3037.13    90.6 3032.88   110.8 3026.96   159.2  3017.2
     240 3017.48   304.5 3019.14   316.6 3020.55   341.2 3019.21   348.9 3017.62
   362.5 3012.36   394.5 3014.21   405.4 3012.67   444.3 3013.62   472.8 3012.02
   490.2 3011.04   497.6 3012.01   514.4 3013.89   530.6 3013.97   546.8 3016.33
   567.4 3012.44   587.7 3014.59   597.8 3019.98   616.3 3034.17   631.5  3043.4
     649 3045.97   657.2 3050.98   665.8 3053.89     694 3068.69   713.3 3076.64
#Mann= 6 ,-1,0
       0      .1       0     340     .08       0     440     .06       0
   472.8    .045       0   497.6     .06       0  633.64      .1       0
#XS Ineff= 2 , 0
          230.19 3022.22
Permanent Ineff=
       F       F
Bank Sta=472.8,497.6
XS Rating Curve= 0 ,0
Exp/Cntr=0.3,0.1

Type RM Length L Ch R = 1 ,147549  ,254.6,254.6,254.6
XS GIS Cut Line= 3
2346326.27376559  642553.50098222346689.72424426642366.819599977
2346897.88224568642213.179170359
#Sta/Elev= 30
       0 3058.91    20.1 3050.11    29.1  3048.1    56.1 3035.41    87.8 3024.22
   105.6 3019.56   132.4 3016.86   144.3    3014   191.8 3013.74   222.5  3016.3
     245 3016.73     263 3016.29   283.9 3012.91   339.4 3016.05   384.4 3013.81
   421.6 3014.92   431.4 3012.74   451.4 3012.46   458.5 3011.16   498.9 3010.09
   508.8 3011.12     531 3012.67   559.5 3009.95   583.3 3018.86   593.2    3027
   608.9 3034.31   620.4 3036.02   631.8 3042.45   655.2 3051.93   667.3 3054.79
#Mann= 5 ,-1,0
       0      .1       0  428.59     .06       0   458.5    .045       0
   508.8     .06       0  548.59      .1       0
#XS Ineff= 2 , 0
          243.75 3023.22
Permanent Ineff=
       F       F
Bank Sta=458.5,508.8
XS Rating Curve= 0 ,0
Exp/Cntr(USF)=0,0
Exp/Cntr=0.3,0.1

Type RM Length L Ch R = 1 ,147294  ,220.3,220.3,220.3
XS GIS Cut Line= 3
2346442.26059355642800.5867217722346836.82959355642577.490462092
2347048.33520566642403.302219338
#Sta/Elev= 30
       0 3055.09      16 3049.79    80.1 3036.79    94.1 3030.95   122.9  3013.2
   130.1  3010.7     163 3010.65   177.1 3014.08   213.6 3012.44     232 3014.92
   291.7 3015.22   310.1  3011.4   376.7 3012.84   397.4  3010.8   411.2 3012.57
   432.5 3012.98   457.6  3011.9   473.2  3008.2     490  3010.6   504.9 3010.91
   541.9 3008.67   587.2 3007.64   595.1 3008.72   611.1 3015.79   623.4 3018.32
   632.1  3023.3     639 3024.22   648.8 3028.64   661.4 3031.99   727.3 3060.27
#Mann= 5 ,-1,0
       0      .1       0   541.9    .045       0   595.1      .1       0
  663.27     .06       0  683.27      .1       0
#XS Ineff= 2 , 0
          181.35 3018.73
Permanent Ineff=
       F       F
Bank Sta=541.9,595.1
XS Rating Curve= 0 ,0
Exp/Cntr=0.3,0.1

Type RM Length L Ch R = 1 ,147074  ,409.4,409.4,409.4
XS GIS Cut Line= 3
2346561.21921501643101.6034716982346920.83778894642814.609959284
2347149.56557087642588.986642997
#Sta/Elev= 30
       0 3099.87      55 3072.68    96.9 3055.23   109.7  3052.3     139 3040.37
   170.3 3030.45     188 3020.79   210.2 3011.79   252.9 3008.65   264.3 3011.42
   285.3 3010.99   301.3 3007.61   346.7 3006.84   382.5 3008.92   418.3 3007.17
   429.3 3010.19   464.8 3011.42   500.2 3010.37     521 3006.45     554 3008.78
   582.3 3007.02   604.9 3010.09630.36773008.092   638.7 3006.74  681.74 3008.11
   695.7 3017.16   712.4 3015.71   723.2 3019.72   743.5 3022.68   781.4 3037.86
#Mann= 4 ,-1,0
       0      .1       0630.3677    .045       0  681.74      .1       0
   710.1     .06       0
#XS Ineff= 2 , 0
          182.05  3017.2
Permanent Ineff=
       F       F
Bank Sta=630.3677,681.74
XS Rating Curve= 0 ,0
Exp/Cntr(USF)=0,0
Exp/Cntr=0.3,0.1

Type RM Length L Ch R = 1 ,146665  ,114.8,114.8,114.8
XS GIS Cut Line= 2
2346745.87712732  643236.04563862347336.20969589642764.306491119
#Sta/Elev= 30
       0 3083.38    52.1 3058.07    79.7 3040.25    97.6 3031.52   115.6 3017.89
   126.3 3012.18   136.1  3008.9   194.4 3009.52   222.8 3007.39   248.7  3007.5
   262.7 3005.28     274 3008.76   279.4 3009.14   335.8 3009.19   353.7  3008.4
     385 3004.44   395.4 3003.17  424.07 3004.48   456.2 3004.46   468.9 3005.62
   484.2    3004   571.3 3008.32     590 3005.37   604.2 3006.61   648.1 3007.07
   663.9 3011.14   678.8 3022.73   696.6 3029.59   722.2 3032.53   755.7 3042.43
#Mann= 5 ,-1,0
       0      .1       0     385    .045       0  424.07      .1       0
     580     .06       0     700      .1       0
Bank Sta=385,424.07
XS Rating Curve= 0 ,0
Exp/Cntr=0.3,0.1

Type RM Length L Ch R = 1 ,146550  ,262.4,262.4,262.4
XS GIS Cut Line= 3
2346798.61211392643366.6045029452347028.06317368643150.002702529
2347391.51365235642874.661430813
#Sta/Elev= 30
       0 3107.35    19.1 3097.28    84.2 3068.93    95.3 3061.77   106.7 3058.42
   130.3  3046.2   177.5 3014.26   194.5 3006.82   222.2 3007.83   244.2 3004.55
   304.9 3007.21   345.8 3005.34   376.5 3009.26     419  3007.8   433.3 3003.63
   447.5 3002.48   469.3  3003.6   484.7 3005.89   547.5 3002.42   556.6 3005.92
   564.6 3006.23   591.7 3003.42   611.8 3006.21   626.8 3004.76   681.7  3005.2
   693.1 3010.56   707.4 3013.17   715.9 3019.57   737.2 3027.53   771.5 3038.15
#Mann= 5 ,-1,0
       0      .1       0   433.3    .045       0   469.3      .1       0
  655.54     .06       0  771.51      .1       0
#XS Ineff= 2 , 0
          222.82 3019.55
Permanent Ineff=
       F       F
Bank Sta=433.3,469.3
XS Rating Curve= 0 ,0
Exp/Cntr(USF)=0,0
Exp/Cntr=0.3,0.1

Type RM Length L Ch R = 1 ,146287  ,262,262,262
XS GIS Cut Line= 2
2347001.82220072643607.1152080122347556.00531363 642986.78741487
#Sta/Elev= 30
       0 3111.73    45.6 3095.64   123.6 3057.74   152.8 3045.71   192.8 3026.47
   231.7 3012.12     241 3007.14   283.5 3001.58   297.7 3003.25   321.7  3002.3
   372.7 3004.75   405.8 3002.08   435.8 3003.77   459.8 3001.87     496 3000.53
   515.8 3001.86   531.9 3004.48   561.1 3002.03   603.9 3004.44   624.8 3001.15
   640.9 3002.71   668.8  3001.7   678.4 3004.06   694.5 3011.33   699.9 3012.37
     712 3011.41   726.7 3020.28   758.9 3031.33     790 3044.19   831.8 3064.77
#Mann= 5 ,-1,0
       0      .1       0   459.8    .045       0   515.8      .1       0
     650     .06       0     790      .1       0
Bank Sta=459.8,515.8
XS Rating Curve= 0 ,0
Exp/Cntr=0.3,0.1
